HEC-RAS study GSCR.prj: GSCR

--- GSCR.g01 (geometry) --- (continued)

Type RM Length L Ch R = 1 ,68079.7 ,489.4,479.5,464.9
XS GIS Cut Line= 3
     1480872.434      263319.995     1479214.691      263470.699
     1478145.871       263619.04
#Sta/Elev= 30
       0     996    88.1  988.97   205.6   965.7   254.6  945.06   342.7  898.22
   450.4  865.86   538.5  861.25   607.1  865.21   724.6  882.48   812.7  878.26
   969.4  837.23  1135.8   803.1    1224  791.24  1351.2  780.35  1429.6  798.64
  1498.1  809.78  1576.4  802.46    1596  796.49  1664.6  762.47  1713.6  732.69
  1782.3  711.05  1968.7  710.24  2213.9  702.27  2243.4   701.8    2312  701.84
  2390.5  708.95  2429.7  733.42  2439.5  737.32  2508.2  751.19  2743.6  779.63
#Mann= 3 , 0 , 0
       0      .1       0  2213.9    .045       0    2312     .06       0
Bank Sta=2213.9,2312
XS Rating Curve= 0 ,0
Exp/Cntr=0.3,0.1

Type RM Length L Ch R = 1 ,67600.2 ,854.2,841.2,827.6
XS GIS Cut Line= 3
     1479388.059      261971.037     1479143.267      262627.287
     1478037.364      263493.172
#Sta/Elev= 30
       0  937.71    68.1  937.41    97.3  935.21   272.4  908.06   418.3  894.64
     467  884.82     574  871.25   612.9   863.5   651.8  851.66   749.5  831.45
   818.3  796.92   847.8  777.89     887  747.89   916.5  734.49     946     726
  1250.5  702.92  1309.4  705.13  1574.6  707.74  1605.7705.6655  1623.7  700.89
  1633.5  700.62  1653.2  701.86    1663  704.65  1672.8  708.16  1702.3   725.5
  1712.1  728.42  1859.4  738.69  1987.1  750.81    2046  759.93    2105  772.12
#Mann= 3 , 0 , 0
       0     .06       0  1605.7    .045       0    1663      .1       0
Bank Sta=1605.7,1663
XS Rating Curve= 0 ,0
Exp/Cntr=0.3,0.1

Type RM Length L Ch R = 1 ,66759   ,812.5,830,847
XS GIS Cut Line= 2
      1477999.17      262197.165     1477572.086      263467.999
#Sta/Elev= 30
       0  876.95    39.1  871.34    88.1  860.14   127.2  848.44   264.2  803.23
   303.4  788.66   342.5  770.93   362.1  765.02   391.4  759.81     411  753.52
   459.9  729.18   489.3  712.44   499.1  708.04   518.7  702.61   538.2   700.6
   577.4   700.6   587.2  701.55   606.7  704.17     685  706.26   949.2  709.15
   988.4  710.58  1017.7   720.1  1037.3  723.57  1047.1  727.44  1135.2  769.89
  1203.7  807.65  1223.2  817.59  1301.5  851.22  1321.1  858.84  1340.7  864.98
#Mann= 3 , 0 , 0
       0      .1       0   518.7    .045       0   587.2     .06       0
Bank Sta=518.7,587.2
XS Rating Curve= 0 ,0
Exp/Cntr=0.3,0.1

Type RM Length L Ch R = 1 ,65928.9 ,835.7,810.1,783.8
XS GIS Cut Line= 3
     1477806.461      261988.832     1476941.878      262447.165
      1476811.67      263035.707
#Sta/Elev= 30
       0  876.97    78.3  867.56   176.1  852.03   195.7  847.93   225.1  838.91
   244.6  831.44   313.1  790.29   371.8  759.27   499.1  709.35   518.6  706.48
   636.1  700.68   655.6  699.88   694.8  701.38   733.9  710.08   743.7  714.51
   782.8  745.58   802.4  756.58   900.3  785.49   939.4  788.31   968.8  792.32
     998  792.47  1114.7  783.24  1143.8   777.3    1173  767.61  1182.7  770.04
  1221.6  785.29  1231.3  787.58  1289.7  794.08  1474.4  806.43  1581.3   811.5
#Mann= 3 , 0 , 0
       0     .06       0   636.1    .045       0   694.8     .06       0
Bank Sta=636.1,694.8
XS Rating Curve= 0 ,0
Exp/Cntr=0.3,0.1

Type RM Length L Ch R = 1 ,65118.9 ,635.8,639.8,643.4
XS GIS Cut Line= 4
     1476822.086      261384.665     1476634.586      261764.874
     1476681.461      262514.874     1476473.128      262952.374
#Sta/Elev= 30
       0  945.79    38.5  936.49    57.8  928.68   115.6  911.35   173.4  898.82
   250.5  877.74     289  866.02     318   858.8   337.2  851.89     395  812.68
   423.9   795.1     463  769.18   492.2  754.01   550.8  714.26   570.3  702.38
   580.1  700.05   589.8   699.7   628.9  700.39   911.9  718.43  1009.5  726.92
  1058.3  728.11  1204.5  726.23  1262.6  726.94  1301.4  732.01  1398.3  741.03
  1495.2  756.67    1534  767.06  1572.7  782.39  1582.4  785.27    1660  804.02
#Mann= 3 , 0 , 0
       0     .06       0   570.3    .045       0   628.9      .1       0
Bank Sta=570.3,628.9
XS Rating Curve= 0 ,0
Exp/Cntr=0.3,0.1

Type RM Length L Ch R = 1 ,64479   ,693.2,717.5,740.4
XS GIS Cut Line= 3
     1476296.045      261395.082     1476040.836      261749.249
     1475957.503      262686.749
#Sta/Elev= 30
       0  859.85    77.6  840.03   116.4  832.23   310.4  787.54   436.5  757.11
   534.6  734.95     613  716.19   681.6  701.68   701.2  699.98   730.7   699.7
   750.3  700.24   838.5  709.17   877.7  711.58   887.5   712.9   897.3  715.25
   946.4  729.41   985.6   739.5    1015  749.04  1034.6  757.78  1054.2  768.62
    1064  774.82  1103.2  802.52    1113  808.44  1211.1  854.22  1250.3   870.9
  1279.7  880.53  1299.3  885.03  1309.1  885.93  1318.9  885.86  1377.7  884.19
#Mann= 3 , 0 , 0
       0      .1       0   681.6    .045       0   750.3     .06       0
Bank Sta=681.6,750.3
XS Rating Curve= 0 ,0
Exp/Cntr=0.3,0.1

Type RM Length L Ch R = 1 ,63761.6 ,537.6,537.7,536.6
XS GIS Cut Line= 3
      1476155.42       261337.79     1475363.753      261691.957
     1475259.586      262301.332
#Sta/Elev= 30
       0  842.14    68.2  825.84   136.4  811.92   204.6  796.11   292.3  777.01
     380  751.78   448.3  737.59   467.8  731.17   506.7  716.26     536  711.92
   652.9  699.52   662.6   699.3   701.6  699.54   711.4  700.35   730.8  705.68
   750.3  708.83   760.1  712.14   808.8  742.12   857.5   768.8   867.3  773.25
   916.3  787.11   975.2  801.14  1073.4   820.9  1083.2  821.93  1122.4  821.56
  1220.5  825.21  1240.2  827.82  1289.2  840.84  1308.9  843.82  1485.5   856.4
#Mann= 3 , 0 , 0
       0      .1       0   652.9    .045       0   711.4     .06       0
Bank Sta=652.9,711.4
XS Rating Curve= 0 ,0
Exp/Cntr=0.3,0.1

Type RM Length L Ch R = 1 ,63223.8 ,415.8,418,420.3
XS GIS Cut Line= 3
     1475983.545       260931.54     1475072.086      261358.624
     1474775.211      261723.207
#Sta/Elev= 30
       0  854.34    78.2  848.61   166.1  838.86   185.7  833.84   224.8  820.86
   263.8  809.83   361.6  776.89   410.4  752.85   420.2  746.85     430  739.12
   459.3  711.28   469.1  703.01  472.96701.2909   478.8  698.69   488.6   698.2
   527.7  698.56   547.2  701.14   625.4  703.93   654.8  706.07   723.2  706.34
   752.5   708.2     772  714.59   869.7   754.6   957.7   783.8  1016.4  790.81
  1104.5  808.75  1192.7  818.64  1241.6  830.79  1310.2  840.24  1476.7  850.08
#Mann= 3 , 0 , 0
       0     .08       0  472.96    .045       0   547.2      .1       0
Bank Sta=472.96,547.2
XS Rating Curve= 0 ,0
Exp/Cntr=0.3,0.1

Type RM Length L Ch R = 1 ,62805.9 ,614.9,617.4,619.5
XS GIS Cut Line= 2
     1475837.711      260592.999     1474712.711      260988.832
#Sta/Elev= 30
       0  832.59    58.6  841.19    78.2  842.57   136.9  842.91   166.2  841.33
   185.7  838.99   205.3  834.24   215.1  831.32   234.6  823.14     391  747.38
   420.3  731.32   469.2  701.02     479  698.07   488.8  697.42   520.9698.4572
   557.2  703.49   615.8  706.26   645.2  709.98   684.3  713.48   703.8  716.72
   723.4  722.54   762.5  736.38   938.4  805.47   987.3  822.15  1036.2  840.43
  1055.8   845.8  1094.8  853.82  1153.5  867.09  1173.1  870.87  1192.6  873.64
#Mann= 3 , 0 , 0
       0     .06       0   469.2    .045       0   520.9      .1       0
Bank Sta=469.2,520.9
XS Rating Curve= 0 ,0
Exp/Cntr=0.3,0.1

Type RM Length L Ch R = 1 ,62188.5 ,907.4,923.4,938.9
XS GIS Cut Line= 2
     1475764.795      260046.124     1474493.961      260348.207
#Sta/Elev= 30
       0  787.29    39.3  783.44     108  770.88   235.7  740.98   245.5  740.61
   255.4  742.62   284.8  756.96   304.5  761.75   353.6  761.37     383  758.98
   402.7  753.89   432.1   738.9     442  735.21   530.4  706.65   608.9  703.42
   628.6  700.25   648.2  696.81   667.8   696.6   687.5  697.44   697.3  699.72
   736.6  710.21   766.1  713.84     825  738.94   883.9  758.65   972.3  782.61
  1149.1  842.33    1208  853.18  1227.7  858.56  1276.8  879.12  1306.2  889.68
#Mann= 3 , 0 , 0
       0     .06       0   628.6    .045       0   697.3      .1       0
Bank Sta=628.6,697.3
XS Rating Curve= 0 ,0
Exp/Cntr=0.3,0.1

Type RM Length L Ch R = 1 ,61265.1 ,463.3,460,456.7
XS GIS Cut Line= 2
     1475759.586      259577.374     1474947.086      259176.332
#Sta/Elev= 30
       0  806.74    48.7  802.87    68.2  802.53    77.9  801.18   116.9  791.61
   194.9  775.27   272.8     751   331.3   731.3   350.7  726.08     380  719.58
   457.9   707.6   584.6  695.93   613.8   694.8   633.3  694.85     643  695.83
   648.2697.6925   652.8  699.34   672.3  710.74   711.2  737.66   730.7  749.37
   740.5  753.16   759.9  757.22   769.7  762.87   808.7  790.78   837.9  816.97
   847.6  824.42   857.4  828.84   876.9   834.9   896.3  832.17   906.1   831.6
#Mann= 3 , 0 , 0
       0      .1       0   584.6    .045       0   648.2     .08       0
Bank Sta=584.6,648.2
XS Rating Curve= 0 ,0
Exp/Cntr=0.3,0.1

Type RM Length L Ch R = 1 ,60805.1 ,712.8,665.1,616.6
XS GIS Cut Line= 3
     1476242.225      259158.537      1475257.85      258840.828
     1474988.753      259103.415
#Sta/Elev= 30
       0  836.37    48.8  844.32   165.9  867.25   204.9  871.48   234.2  870.43
   263.5  862.92   331.8  839.83   361.1  827.05   478.2  770.75   585.5  727.57
     605  721.06   624.5  716.76   653.8  712.46   751.4  705.77   839.2  696.21
   868.5   694.8   907.5  695.76   917.3  699.97   936.8   711.7   956.3     716
   975.8  716.46  1034.4  712.58  1111.5   718.8  1150.1  724.48  1256.1  746.19
  1275.4  747.83    1285  749.86  1323.6  766.58  1371.8  778.58  1410.4  796.82
#Mann= 3 , 0 , 0
       0      .1       0   839.2    .045       0   917.3      .1       0
Bank Sta=839.2,917.3
XS Rating Curve= 0 ,0
Exp/Cntr=0.3,0.1

Type RM Length L Ch R = 1 ,60140   ,445.4,467,487.7
XS GIS Cut Line= 5
     1475455.767      258111.662     1475073.506      258552.511
     1475145.003      258874.249     1474983.545      259061.749
      1474936.67      259092.999
#Sta/Elev= 30
       0  813.58    29.2  825.88    48.6  831.84    68.1  833.76   145.9  836.12
   233.4  822.81   350.1  817.39   398.7  816.71   447.4  810.03   486.2  799.88
   534.9  796.52   554.3  791.73   593.2  777.22   602.9  769.39   622.3  747.05
     632  737.61   651.4  720.94     661  714.51   670.7  710.17   709.5  696.88
   728.9  694.11   748.3  694.54   767.7  699.02   796.8  705.05   951.2  718.34
  1017.8   732.3  1046.3  740.73  1074.9  744.15  1122.4  763.71  1216.9  796.65
#Mann= 3 , 0 , 0
       0      .1       0   709.5    .045       0   767.7     .08       0
Bank Sta=709.5,767.7
XS Rating Curve= 0 ,0
Exp/Cntr=0.3,0.1

Type RM Length L Ch R = 1 ,59673   ,586.5,594.5,602
XS GIS Cut Line= 2
     1474983.545      258353.415      1474342.92       259087.79
#Sta/Elev= 30
       0  792.34      39  789.88    48.7  788.71    68.2  784.46   107.2   773.5
   175.4  750.36   263.1  724.83   302.1  714.67   438.5  704.66   448.3  703.53
     458  701.14   467.8  697.58   477.5  694.55   487.3   693.2   516.5  693.31
   526.2   694.1     536  697.03   555.5  705.76   565.2  708.86   584.7   712.5
   604.2  722.42   662.7  757.42   750.4  812.84   760.1  819.38   779.6  835.08
   789.4  841.67   799.1  845.72   838.1  855.21   857.6  857.63   974.5  856.27
#Mann= 3 , 0 , 0
       0      .1       0   467.8    .045       0     536      .1       0
Bank Sta=467.8,536
XS Rating Curve= 0 ,0
Exp/Cntr=0.3,0.1

Type RM Length L Ch R = 1 ,59078.5 ,613.2,609.2,604.7
XS GIS Cut Line= 2
      1474749.17       258056.54     1473952.295       258494.04
#Sta/Elev= 30
       0  817.96    19.6  814.86    29.3  812.72    39.1  809.55    58.6  802.34
    97.8  789.71     176  760.59   224.8  740.26   244.4  730.14   293.2  702.59
   307.7695.9954   312.8   694.2   322.6   693.2   357.7693.5123   508.3  710.94
   518.1  712.19   527.8  714.88   547.4  722.55     567  731.55   576.7  737.15
     606  756.24   625.6  765.91   674.5  782.46   713.6  797.34   742.9  806.82
   791.8  819.59   821.1  829.26   879.8  845.39   889.5  847.72   909.1  850.53
#Mann= 3 , 0 , 0
       0      .1       0   307.7    .045       0   357.7      .1       0
Bank Sta=307.7,357.7
XS Rating Curve= 0 ,0
Exp/Cntr=0.3,0.1

Type RM Length L Ch R = 1 ,58469.3 ,422.4,424.7,427
XS GIS Cut Line= 2
     1474353.336      257520.082     1473733.545      258030.499
#Sta/Elev= 30
       0  784.62    39.2  784.91    58.8  784.18   137.1   776.6   146.9   774.4
   156.7  770.94   195.8  754.03     235   741.6   244.8  738.23   254.6  733.89
   274.2   723.8     284  717.82   303.5  703.46   313.3  697.25   323.1  693.63
     341   693.2   362.3  693.61   372.1  694.71   499.4  713.74   509.2   716.4
     519  720.11   577.7  743.85   587.5  747.07   597.3  749.05   607.1   750.2
   646.2  749.82   695.2   751.4   734.4  753.97   773.5  757.47   802.9  758.84
#Mann= 3 , 0 , 0
       0      .1       0   313.3    .045       0   372.1      .1       0
Bank Sta=313.3,372.1
XS Rating Curve= 0 ,0
Exp/Cntr=0.3,0.1

Type RM Length L Ch R = 1 ,58044.6 ,486.8,492.1,497.4
XS GIS Cut Line= 3
     1475033.892      257606.453     1474035.628      257270.082
      1473436.67      257665.915
#Sta/Elev= 30
       0  782.62    87.8  771.73   107.3  766.78   156.1  750.11   204.8  743.29
   214.6  743.41   224.3  746.96   243.8  759.18   263.4  766.78   302.4  773.27
   380.4  781.71   477.9   773.3     556  763.73   682.8  774.69   770.6  775.49
   907.1  769.97  1053.4  761.24  1102.6  762.01  1132.1  753.84  1191.1  726.61
  1240.3  696.86  1250.1  693.84  1269.8   693.2  1299.3  693.64  1407.5  704.67
    1437  715.05  1535.3   735.7  1594.3  746.58  1653.3  755.13  1771.4  776.77
#Mann= 3 , 0 , 0
       0      .1       0  1240.3    .045       0  1299.3      .1       0
Bank Sta=1240.3,1299.3
XS Rating Curve= 0 ,0
Exp/Cntr=0.3,0.1

Type RM Length L Ch R = 1 ,57552.4 ,687.4,693.9,699.6
XS GIS Cut Line= 3
     1475489.838       256756.41     1474187.755       256756.41
     1473041.921      257178.285
#Sta/Elev= 30
       0  892.92   166.4  860.59   362.2  804.61   548.2   736.1   616.8  718.88
   646.2  715.23   695.1  711.38   724.5  714.64     744  719.96   812.6  750.23
   881.1  760.74  1067.1  770.66  1243.3  784.77  1311.8  775.36  1399.8  744.62
  1429.1     731  1487.7  721.41  1565.8  693.07  1800.3  700.61  1819.8  703.07
  1849.1  712.87  1858.9  712.72    1898  696.11    1937   691.8  1976.1  693.47
  2103.1  708.82  2210.5  756.93  2298.4  791.09    2445   775.2  2523.1  772.52
#Mann= 3 , 0 , 0
       0      .1       0    1898    .045       0  1976.1      .1       0
#XS Ineff= 2 , 0
         1851.13   724.4
Permanent Ineff=
       F       F
Bank Sta=1898,1976.1
XS Rating Curve= 0 ,0
Exp/Cntr=0.3,0.1

Type RM Length L Ch R = 1 ,56858.6 ,700.2,707.9,714.7
XS GIS Cut Line= 3
      1474953.38      255574.118      1473765.88      256360.577
     1473067.963      256417.868
#Sta/Elev= 30
       0  839.61    98.2  835.94   186.6  813.98   255.4  808.68   343.8   807.1
   392.9  810.21   628.7  809.36   746.5  814.57   834.9  822.05   913.5  816.43
  1021.6  819.46    1051  815.64  1168.9  790.69  1306.4  785.81  1345.7  780.67
  1394.8  766.37    1434   750.2  1482.7  734.93  1521.6  718.14  1560.5   717.5
  1609.1  706.54  1696.6  698.58  1871.7   690.2  1900.9  689.45  1920.3  689.65
  1939.8  694.73  2017.6  744.93    2076  776.67  2095.4   784.8  2124.6  787.71
#Mann= 3 , 0 , 0
       0      .1       0  1871.7    .045       0  1939.8      .1       0
Bank Sta=1871.7,1939.8
XS Rating Curve= 0 ,0
Exp/Cntr=0.3,0.1

Type RM Length L Ch R = 1 ,56150.7 ,494.4,459.2,423.3
XS GIS Cut Line= 2
     1474166.921      255923.077     1473146.088      255678.285
#Sta/Elev= 30
       0   829.6    29.4  821.24      49  815.13    88.3   800.8   196.2  773.61
   215.8  769.38   402.2  732.31   500.4   715.4     520  712.27   529.8  711.18
   667.2  699.14   686.8  698.19   735.8  698.98   794.7  697.57   804.5  696.32
   814.3  693.53   824.1  690.37   833.9  688.63   843.7   688.6   863.4  688.68
   870.1 692.365   873.2  694.07   892.8  711.52   902.6  718.26   912.4  723.35
   922.2  727.45     932  729.42   941.8   729.8   981.1  729.24  1049.8  726.94
#Mann= 3 , 0 , 0
       0      .1       0   814.3    .045       0   870.1      .1       0
Bank Sta=814.3,870.1
XS Rating Curve= 0 ,0
Exp/Cntr=0.3,0.1

Type RM Length L Ch R = 1 ,55691.5 ,411.7,403.9,396.3
XS GIS Cut Line= 3
     1473489.838      254870.993     1473317.963      255563.702
     1473146.088      255641.827
#Sta/Elev= 30
       0  884.63    29.3   882.9    68.4  879.02   136.9  875.89     176   872.5
   195.5   869.9   205.3  867.57   224.9  860.18   254.2  845.12   293.3  822.64
   303.1   816.1   322.6   799.9   391.1  739.09     440  698.57   446.2 694.409
   449.7  692.06   459.5  688.94   469.3   688.5   488.8  688.66   498.6  689.72
   518.2  694.95     528  697.17   547.5   699.3   625.7  702.72   664.8  705.87
   713.7  713.92   808.1  725.45     827  726.13   855.3  724.08   902.5  722.61
#Mann= 3 , 0 , 0
       0      .1       0   446.2    .045       0   518.2      .1       0
Bank Sta=446.2,518.2
XS Rating Curve= 0 ,0
Exp/Cntr=0.3,0.1

Type RM Length L Ch R = 1 ,55287.6 ,592,573.7,555.1
XS GIS Cut Line= 3
     1472928.591       254825.26     1473019.736      255745.399
     1472937.271      257242.795
#Sta/Elev= 30
       0  894.99    78.7  892.23   108.2  888.61   147.6  879.78   196.7  863.29
   334.4  830.01   344.3  823.38   383.6  784.13   452.5  724.02   479.8694.1504
   491.8  688.76   501.7   688.5     541  688.86   550.8  691.49   609.9   700.1
   786.9  705.13   875.5  715.05   944.2  713.09   963.8  716.48   993.2  725.73
  1257.9   729.8  1297.1  732.65  1434.3   746.5  1532.4  759.57    1748   808.3
  1855.8  817.27  1924.4  818.69  2179.3  786.14  2365.5  778.14  2424.3  768.51
#Mann= 3 , 0 , 0
       0      .1       0   479.8    .045       0   550.8      .1       0
Bank Sta=479.8,550.8
XS Rating Curve= 0 ,0
Exp/Cntr=0.3,0.1

Type RM Length L Ch R = 1 ,54713.9 ,971.6,1010.3,1047.8
XS GIS Cut Line= 6
     1472781.505      254959.535     1472474.213      255652.243
     1472927.781      256002.523     1472854.806      257238.454
     1472390.396      258614.322     1473445.084      260888.628
#Sta/Elev= 30
       0  864.65   177.2  822.21   472.4  777.66   541.3  719.48   570.8  710.28
   679.1  757.22   777.2  759.24   931.1690.1602   963.6  688.31   990.9  690.83
  1330.9  725.44  1714.1  747.78  1940.1  785.68  2087.5  787.16  2382.3  767.98
    2726  780.68  2863.3     772  3187.1  791.04    3295  839.42  3589.4  891.46
  3981.9 1018.13  4483.2 1045.26  4650.3 1076.69  4797.8 1072.59  5023.9 1013.57
  5387.6 1027.88  5702.2 1005.43  5977.5 1017.81  6164.3 1050.04  6528.1 1074.58
#Mann= 3 , 0 , 0
       0      .1       0   931.1    .045       0   990.9      .1       0
Bank Sta=931.1,990.9
XS Rating Curve= 0 ,0
Exp/Cntr=0.3,0.1

Type RM Length L Ch R = 1 ,53703.6 ,837,860.6,883.9
XS GIS Cut Line= 6
     1472754.111      254929.426     1472423.382      255614.322
     1472038.052      256233.246     1471287.966      257103.906
     1470788.834      257407.725     1469512.792      259868.663
#Sta/Elev= 30
       0  863.38   243.8  807.19   497.3  767.19     585  711.22   702.1  751.13
   760.6   753.8   837.7  742.95   905.2  711.31  1051.1  695.96  1560.9  689.21
  1580.5   687.7  1659.1   688.9  1757.3  713.68  1835.9  711.21  1904.6  743.59
    2052  782.64  2543.1  866.33  2651.1  897.87  3304.3  994.14  4031.7 1004.96
  4159.5   980.7  4267.6  989.04  4375.8  977.69  4542.9  941.67  4611.7  951.37
  4719.8   988.9  4877.1 1005.25    5575 1005.58  5830.6    1044  6007.6 1052.94
#Mann= 3 , 0 , 0
       0      .1       0  1560.9    .045       0  1659.1      .1       0
Bank Sta=1560.9,1659.1
XS Rating Curve= 0 ,0
Exp/Cntr=0.3,0.1

Type RM Length L Ch R = 1 ,52843   ,218.5,219.7,220.7
XS GIS Cut Line= 4
     1472713.796      254923.077     1472385.671      255532.452
     1471739.838      255428.285     1470791.707      257344.936
#Sta/Elev= 30
       0  856.44   253.4  798.02   506.9  751.88   555.6   716.2   575.1  710.78
   692.1  736.37   789.7  708.61     819  693.19   848.3   687.7   879.5 688.919
    1112   704.2  1346.3  747.49  1405.1  765.91  1571.9  792.81  1836.7  814.87
  2101.6  849.54    2131   847.3  2268.3   807.1  2405.6  838.98  2513.5  820.74
  2572.4  797.14  2641.1     840  2768.6  877.34    2847  882.64  2954.9  841.74
  3043.2  887.26  3151.1  887.54  3219.8  926.56  3268.8  944.98  3484.6  983.09
#Mann= 3 , 0 , 0
       0      .1       0     819    .045       0   879.5     .06       0
Bank Sta=819,879.5
XS Rating Curve= 0 ,0
Exp/Cntr=0.3,0.1

Type RM Length L Ch R = 1 ,52623.3 ,963.7,932.4,901.1
XS GIS Cut Line= 3
     1472666.921       254912.66     1472427.338      255324.118
     1471786.713       255193.91
#Sta/Elev= 30
       0  847.74      68  830.41   106.9  822.95   194.3   803.1   349.8   770.2
   417.8  754.15   456.7  742.15   476.1  738.11   534.7  719.39   573.7   705.4
     603  693.26   612.9690.2477   632.2  687.66   651.8   686.8   661.5  686.96
   671.3  687.98     681  690.07   700.5  692.25   788.4  697.51   817.6  698.69
   856.6  698.66   905.4  695.56     925  696.03   944.5  697.67   954.2   699.4
   993.2  709.32  1022.5  714.27  1071.3  719.25  1090.8  719.92  1129.8  719.68
#Mann= 3 , 0 , 0
       0      .1       0   612.9    .045       0     681     .06       0
Bank Sta=612.9,681
XS Rating Curve= 0 ,0
Exp/Cntr=0.3,0.1

Type RM Length L Ch R = 1 ,51690.9 ,1034.8,1000,962.7
XS GIS Cut Line= 4
      1472890.88      253495.993     1472099.213      254074.118
     1471786.713       254818.91     1471791.921       255131.41
#Sta/Elev= 30
       0  934.98   107.8  920.15   205.9  912.01   254.9     910   313.7  900.26
   372.5  898.63   460.7  882.95   558.8  876.47   656.8  866.04   735.2  847.49
     794  826.93   921.5  774.56  1009.5  741.37  1058.1  710.72  1067.9  707.33
  1126.3   701.9    1282  699.71  1311.2  696.78  1340.3   689.9  1350.1   687.6
  1369.5   686.8  1398.7  686.89  1418.2  690.18    1496  691.19  1612.8  696.21
  1661.5   700.1  1749.1  710.84  2022.4  726.16  2071.2  727.56  2100.5   723.6
#Mann= 3 , 0 , 0
       0     .06       0  1340.3    .045       0  1418.2     .06       0
Bank Sta=1340.3,1418.2
XS Rating Curve= 0 ,0
Exp/Cntr=0.3,0.1

Type RM Length L Ch R = 1 ,50691   ,570.4,592.8,615.2
XS GIS Cut Line= 3
     1471161.713       253475.16      1471265.88       254912.66
     1471760.671      255120.993
#Sta/Elev= 30
       0   958.3    58.8  959.79   127.5  949.64   225.5   947.1   294.1  936.98
     353  931.93   421.6  921.83   598.1  904.94   647.1  897.45   705.9  884.39
   745.2  878.26     804  865.15   862.8  854.82   911.8  839.56   960.8  830.51
  1000.1  829.03  1058.9  835.12  1117.7  837.66  1156.9  821.66  1313.8  774.42
  1470.6  737.55  1538.9  711.55  1577.9  690.17  1587.7  686.41  1626.7   684.2
  1685.3  685.72    1822   696.9  1909.8  717.07  1958.6  723.86  1978.1  724.76
#Mann= 3 , 0 , 0
       0      .1       0  1587.7    .045       0  1685.3     .06       0
Bank Sta=1587.7,1685.3
XS Rating Curve= 0 ,0
Exp/Cntr=0.3,0.1

Type RM Length L Ch R = 1 ,50098.2 ,720.4,738.6,756.1
XS GIS Cut Line= 2
     1470937.755      254501.202      1471297.13      256277.243
#Sta/Elev= 30
       0  827.24   166.5  801.93   372.2   744.8   470.2  745.52   617.1  741.28
   754.2  728.21   832.6  714.84   842.4  707.32   852.2  694.96   861.9  685.26
   881.5   680.4   901.1  683.41   910.9  688.42   930.5   699.2   950.1  702.47
  1008.9  690.44    1195   690.6  1234.1  698.82  1253.7  707.61  1292.9  740.65
  1332.1  768.86  1381.1  796.65  1400.6  803.61  1449.6  813.61  1557.4  858.98
  1606.4  867.59  1635.7  864.55  1782.6  814.05  1792.4  811.66    1812  813.38
#Mann= 3 , 0 , 0
       0      .1       0   852.2    .045       0   910.9      .1       0
#XS Ineff= 2 , 0
                          940.66           704.1
Permanent Ineff=
       F       F
Bank Sta=852.2,910.9
XS Rating Curve= 0 ,0
Exp/Cntr=0.3,0.1

Type RM Length L Ch R = 1 ,49359.6 ,553.7,549.3,545
XS GIS Cut Line= 3
     1470885.671      254532.452      1470265.88      255459.535
     1470088.796      256355.368
#Sta/Elev= 30
       0  815.58   215.2     777   283.7  768.28   430.4  739.44     450  733.66
   479.3  720.07   508.7  715.18   567.4  700.29     763  690.37   802.2  682.32
   831.5   679.9   851.1  679.97   870.6  685.25   890.2   694.4     988  711.45
   997.8  715.42    1076  764.86  1105.4  781.02  1203.6  817.62  1252.6  832.44
  1419.6  864.91  1507.9  876.87  1625.8  879.37  1684.7  885.77  1792.7  891.36
  1822.2  900.31  1881.1  931.47  1920.3  948.27  1979.2  963.78  2028.4  972.69
#Mann= 3 , 0 , 0
       0     .06       0   802.2    .045       0   870.6      .1       0
Bank Sta=802.2,870.6
XS Rating Curve= 0 ,0
Exp/Cntr=0.3,0.1

Type RM Length L Ch R = 1 ,48810.3 ,1220.3,1201.9,1175.5
XS GIS Cut Line= 4
     1470401.296      253860.577     1470161.713      254579.327
     1469786.713      255334.535      1469922.13      256141.827
#Sta/Elev= 30
       0  824.76    39.4  804.68     187  782.99     246  771.15   314.9  777.14
   482.1  809.74     551  819.37   600.2  822.02   639.6  818.22   678.9  809.76
   747.8  784.69   816.5  738.38   885.1  702.44  1022.4  688.03  1051.8  681.21
  1099.8   679.1 1124.69681.9814    1140  685.91  1355.7  693.83  1443.9  705.81
  1571.4  736.27    1669  752.84  1698.3  753.52    1825  740.49  1932.1  745.54
  1971.1  758.69  2058.8  798.22    2205  832.81  2331.7  870.66  2419.4  884.42
#Mann= 3 , 0 , 0
       0     .06       0  1051.8    .045       0 1124.69     .06       0
Bank Sta=1051.8,1124.69
XS Rating Curve= 0 ,0
Exp/Cntr=0.3,0.1

Type RM Length L Ch R = 1 ,47608.4 ,984.6,951.4,918
XS GIS Cut Line= 4
     1467937.755      253699.118      1468828.38      254397.035
     1469474.213      255308.493      1469828.38      255938.702
#Sta/Elev= 30
       0  883.28   108.2  884.01   236.1  843.81   324.7  846.04   432.9  836.27
   521.5  820.23   649.4  819.27   826.5  785.42   924.9  784.23   983.9  770.29
  1111.8     750  1170.7  733.57  1209.9  715.99  1268.7  714.19  1376.5  693.76
  1582.2  684.48  1631.2   679.5  1660.6   678.6  1719.4  680.73  1748.8  687.18
    1886  680.76  2091.8  690.26  2170.2  701.52  2277.9  700.84  2463.5  720.22
  2512.3  731.44  2600.3  740.28  2756.6  766.88    2864  801.97  2971.5  830.94
#Mann= 3 , 0 , 0
       0     .06       0  1631.2    .045       0  1719.4     .06       0
Bank Sta=1631.2,1719.4
XS Rating Curve= 0 ,0
Exp/Cntr=0.3,0.1

Type RM Length L Ch R = 1 ,46657   ,168.3,166.4,165
XS GIS Cut Line= 3
     1468500.255      255730.368     1469161.713      255355.368
     1469536.713      255527.243
#Sta/Elev= 30
       0  732.78    87.7  740.74   126.7  741.75   175.5   740.7     195  736.62
     234  725.36   243.7  720.79   263.2  708.23     273     704   282.7  701.49
   331.4  692.77   341.2  689.52   360.7   680.4   370.4  678.66   380.2   678.6
   419.2  679.12   438.7  681.77   458.2  683.12   575.2  686.56   623.9   686.5
   653.1  687.63   682.4  690.69   740.9  699.77   829.1  700.09   848.8  698.22
   868.4  697.67     947  702.58  1005.9  704.92  1113.9  715.74  1172.9  720.42
#Mann= 3 , 0 , 0
       0      .1       0   360.7    .045       0   419.2     .06       0
Bank Sta=360.7,419.2
XS Rating Curve= 0 ,0
Exp/Cntr=0.3,0.1

Type RM Length L Ch R = 1 ,46490.6 ,353.3,366.6,379.1
XS GIS Cut Line= 3
     1468567.963       255881.41     1469271.088      255464.743
     1469588.796       255631.41
#Sta/Elev= 30
       0  732.63    68.1   734.7   126.5  732.91     146  731.12   155.7  729.38
   175.1  723.45   204.3  710.55   223.8  703.28   243.2  698.57   291.9  690.18
   330.8  680.06   337.9679.0457   350.3   678.6   379.5  678.66   391.2679.7056
   418.4  686.34   437.8  688.21   476.8  689.75   486.5  689.55   515.7  687.29
   525.4  687.29   574.1  689.22     613  691.48   729.7  700.21   768.7  701.96
   817.3  702.25   991.8  715.03  1069.4  719.73  1079.1  720.81  1176.1  736.08
#Mann= 3 , 0 , 0
       0      .1       0   337.9    .045       0   391.2     .06       0
Bank Sta=337.9,391.2
XS Rating Curve= 0 ,0
Exp/Cntr=0.3,0.1

Type RM Length L Ch R = 1 ,46124   ,409.2,410.5,412.4
XS GIS Cut Line= 2
     1468635.671       256068.91      1469453.38      256048.077
#Sta/Elev= 30
       0  736.74    87.6  729.12    97.4  728.09   107.1  726.19   116.8  723.07
   165.5   705.4   175.3  700.57   194.8  686.65   204.5  680.86   214.2  678.77
     224   678.6   272.7  678.61   282.4  679.21   292.1  681.97   301.9  684.63
   311.6  685.49   428.5  686.86   438.2  687.39   447.9  688.73   467.4   692.8
   516.1  704.32   525.8  706.25   545.3  708.98     555  711.06     594  722.45
   613.5  726.59   671.9  736.14   720.6  740.25   740.1   742.7     818   756.3
#Mann= 3 , 0 , 0
       0      .1       0   194.8    .045       0   292.1     .06       0
Bank Sta=194.8,292.1
XS Rating Curve= 0 ,0
Exp/Cntr=0.3,0.1

Type RM Length L Ch R = 1 ,45713.5 ,485.8,517.2,547.4
XS GIS Cut Line= 2
     1468646.088      256454.327     1469583.588      256480.368
#Sta/Elev= 30
       0  722.68    48.8  716.07   146.5  706.27   166.1  703.78   205.2  695.85
   273.5   680.4   283.3  678.74   293.1   678.6   341.9  678.64   351.7  679.09
   361.5  680.51   420.1  690.57   468.9  700.18   498.2   703.5     508   705.3
   517.8     708   527.6  711.55   537.3  713.97   556.9  717.54   576.4  723.23
   625.2   742.6   644.8  749.23   683.9  759.62   742.5  774.15   781.6  788.59
   830.4  808.21   869.5  824.62     889  833.63   918.3  849.06   937.9  857.89
#Mann= 3 , 0 , 0
       0      .1       0   273.5    .045       0   361.5     .06       0
Bank Sta=273.5,361.5
XS Rating Curve= 0 ,0
Exp/Cntr=0.3,0.1

Type RM Length L Ch R = 1 ,45196.3 ,626.7,652.8,676.5
XS GIS Cut Line= 3
     1468625.255      256490.785     1468762.588      257116.002
     1468970.922      258257.495
#Sta/Elev= 30
       0  718.66   155.2  695.94   203.7   680.7   213.4  678.58   232.8     678
   271.6  678.04     291   681.4   310.4   686.9   320.1  687.63   465.5  689.01
   640.1  695.86   728.6  709.46   817.1  719.55   856.5  733.46   895.8  741.25
   964.6  769.62  1013.8  780.07  1023.6  784.57  1033.5  792.02  1053.1  810.29
    1063  817.62  1082.6  828.64  1092.5   832.4    1122  838.96  1230.1  851.08
  1269.5  861.17    1417  871.53  1643.1  881.99  1702.1  886.39  1800.5   886.2
#Mann= 3 , 0 , 0
       0      .1       0   203.7    .045       0     291     .06       0
Bank Sta=203.7,291
XS Rating Curve= 0 ,0
Exp/Cntr=0.3,0.1

Type RM Length L Ch R = 1 ,44543.5 ,426.6,428.7,430.8
XS GIS Cut Line= 2
     1468562.755      256272.035     1467687.755       256975.16
#Sta/Elev= 30
       0  736.03    19.5   736.4      39  734.29   107.4  719.06   136.6  709.31
   165.9  700.89   214.7  695.53   273.3  692.46   302.6  689.39   419.7  689.41
   497.8  687.38   566.1  684.29   575.9  683.52   589.8680.2029   595.4  678.78
   605.2     678   624.7  678.13   634.5  679.76   644.2  684.64     693  721.21
   702.8  727.17   732.1  734.13   780.9   751.9   839.4  770.68   868.7  782.92
   878.5  786.29   888.2  788.24   946.8  789.36  1044.4   783.8  1122.5     776
#Mann= 3 , 0 , 0
       0     .06       0   589.8    .045       0   644.2      .1       0
Bank Sta=589.8,644.2
XS Rating Curve= 0 ,0
Exp/Cntr=0.3,0.1

Type RM Length L Ch R = 1 ,44114.7 ,141.4,144.2,145.8
XS GIS Cut Line= 2
     1468401.296      255933.493     1467531.505      256511.618
#Sta/Elev= 30
       0  718.96   107.4  714.17   214.7  706.83   253.8  707.15   302.6  711.55
   331.9  711.81   380.7  706.69   400.2  701.84   429.5  691.31   439.2  689.54
     488   687.8   614.9  686.84   624.7   685.7   634.4  682.06   644.2  678.44
   663.7     678     693  678.46   702.8  681.52   712.5  684.03   780.9  689.49
   849.2  691.42   858.9  693.47   878.5  706.57   888.2   711.6     898  714.51
   917.5  718.15     937  719.42   976.1  728.83  1015.1  728.84  1044.4  726.76
#Mann= 3 , 0 , 0
       0     .08       0   634.4    .045       0   702.8      .1       0
Bank Sta=634.4,702.8
XS Rating Curve= 0 ,0
Exp/Cntr=0.3,0.1

Type RM Length L Ch R = 1 ,43970.5 ,770.4,747.7,725.9
XS GIS Cut Line= 2
     1468323.171       255881.41      1467390.88      256407.452
#Sta/Elev= 30
       0   711.9    88.4  712.57   117.8  710.98   216.1  710.21   265.2  711.64
   294.6  711.13   314.3  709.36   324.1  707.42   363.4  693.54   373.2  691.38
   392.8  688.92   432.1  687.33   559.8  689.65   589.2     689   618.7  686.47
   628.5   684.8   638.4  681.37   648.2  678.55   667.8     678   697.3  678.34
   705.5680.2477   716.9  685.13   726.7  687.22   746.4  687.34   805.3  690.81
   834.8  693.77   864.2  698.13   883.9  699.71   972.2  701.43  1070.5     700
#Mann= 3 , 0 , 0
       0     .06       0   638.4    .045       0   705.5     .06       0
Bank Sta=638.4,705.5
XS Rating Curve= 0 ,0
Exp/Cntr=0.3,0.1

Type RM Length L Ch R = 1 ,43222.8 ,744.1,721.9,699.7
XS GIS Cut Line= 4
     1467557.546      254777.243     1467338.796      255449.118
     1467250.255      256261.618     1467354.421      256454.327
#Sta/Elev= 30
       0  867.65   127.6  870.09   206.1  876.59   255.2  873.86   284.6  869.83
   323.8  859.82   353.3  859.58   382.7  855.68   559.4  822.48   637.9  814.76
   677.2  808.16   696.8  802.13   803.9  749.56   823.4  734.07   862.3  697.73
   881.7  684.85   891.5   680.2   910.9     676   940.1  676.77   949.8  679.11
   959.6  682.06   969.3   682.8  1173.6  682.85  1368.2  687.93    1378   689.6
  1397.4  697.16  1416.9  702.02  1514.2  706.26  1704.9  699.67    1743  701.96
#Mann= 3 , 0 , 0
       0      .1       0   891.5    .045       0   949.8     .06       0
Bank Sta=891.5,949.8
XS Rating Curve= 0 ,0
Exp/Cntr=0.3,0.1

Type RM Length L Ch R = 1 ,42500.8 ,302.7,330.4,358
XS GIS Cut Line= 4
     1466635.671      255277.243     1466687.755      255980.368
     1467349.213      256532.452     1468567.276      259017.044
#Sta/Elev= 30
       0  831.09      49  835.99   215.4   812.8   440.7  799.83   734.4  720.51
   851.9  680.09   891.1     676   910.7  678.34  1184.8  706.37  1556.8  703.53
  1753.1  740.47  1821.8  762.81  1968.9  778.51  2135.8  757.56  2253.5  771.37
  2371.2  740.58  2469.4  768.07  2665.6  778.86  2753.9   792.5  2793.2  784.16
  2930.6  829.84  2989.4  830.27    3117  861.11  3352.5  939.12  3460.4  951.69
  3715.6  900.63    3902  892.97  4039.4   914.1  4176.7  964.55  4333.7 1004.75
#Mann= 3 , 0 , 0
       0      .1       0   851.9    .045       0   910.7     .06       0
Bank Sta=851.9,910.7
XS Rating Curve= 0 ,0
Exp/Cntr=0.3,0.1

Type RM Length L Ch R = 1 ,42170.4 ,1078.3,1076.3,1073.3
XS GIS Cut Line= 3
      1466578.38      255277.243      1466640.88      256120.993
      1466015.88      257902.243
#Sta/Elev= 30
       0  825.23    49.2  828.11   137.7  812.43   265.6  811.79   462.4  795.05
   619.8  756.68   688.6   727.2   718.2  719.05   836.2  699.96   914.9  695.22
   973.9  679.39   993.5   675.9  1042.7  679.17  1091.9  692.47  1121.4  691.17
  1160.7  682.21  1219.7  683.49  1288.5  702.88  1445.8   719.2  1524.5   734.5
  1652.3  778.09  1740.8  791.03  1799.8   804.8  1868.6   828.3  2084.9  863.39
  2173.4  872.01  2419.2  882.15  2497.8  881.89  2625.6  893.03  2733.8  891.28
#Mann= 3 , 0 , 0
       0     .06       0   973.9    .045       0  1042.7      .1       0
#XS Ineff= 2 , 0
                         1096.51          701.79
Permanent Ineff=
       F       F
Bank Sta=973.9,1042.7
XS Rating Curve= 0 ,0
Exp/Cntr=0.3,0.1

Type RM Length L Ch R = 1 ,41094.1 ,752,750.4,748.3
XS GIS Cut Line= 3
     1466724.213      254933.493      1466078.38      255199.118
     1465849.213      256209.535
#Sta/Elev= 30
       0  788.04    29.5  795.65    39.3  795.26   108.2  781.07   147.5   765.4
   157.4  764.43   216.4  772.32   275.4  775.16   344.2  764.24   422.9  768.06
   481.9  762.47     541  779.54   570.5  782.73   609.8  779.59   698.3  764.56
   747.2  759.93   815.6  757.85   825.4  754.44   854.7  733.54   913.4  679.42
   932.9   674.5   962.2  674.84   981.8  679.56  1177.3  686.84  1294.6  696.74
  1421.6  696.35  1538.9  736.82  1597.6  751.88  1695.3  769.22  1734.4  780.92
#Mann= 3 , 0 , 0
       0      .1       0   913.4    .045       0   981.8     .06       0
Bank Sta=913.4,981.8
XS Rating Curve= 0 ,0
Exp/Cntr=0.3,0.1

Type RM Length L Ch R = 1 ,40343.7 ,778.6,768,755.9
XS GIS Cut Line= 4
     1465646.088      254709.535     1465424.915      255006.627
     1465277.345      256043.953     1465251.304      256291.349
#Sta/Elev= 30
       0  778.17    58.5   765.2   107.2  756.31   214.4  746.78   263.2  732.36
   292.4  727.14   370.4  721.69   468.3  717.93   605.4  701.72   703.3  694.79
   742.5   689.3   781.6  688.74   820.8  684.34   889.4  681.78     909  676.61
   918.8  674.64   948.1     674   977.5  674.07  1006.9  676.27    1046  693.56
  1055.8  695.97  1104.8   696.7  1124.4  699.23  1192.9  723.03  1232.1   734.9
  1261.5  741.75  1339.8   755.1  1418.2  776.81  1485.1  796.69  1666.9  864.25
#Mann= 3 , 0 , 0
       0      .1       0     909    .045       0  1006.9      .1       0
Bank Sta=909,1006.9
XS Rating Curve= 0 ,0
Exp/Cntr=0.3,0.1

Type RM Length L Ch R = 1 ,39575.8 ,649.7,649.7,648.1
XS GIS Cut Line= 2
     1464411.713      254923.077     1464844.005      256048.077
#Sta/Elev= 30
       0  828.65   127.4  794.26   215.6  776.13     245  768.73   284.2   751.4
   323.4  735.91   352.7  719.34   372.3   710.6   382.1  708.73   421.3   713.8
   440.9  712.53   489.9  701.75   548.7  678.72   558.5   675.3   578.1   673.9
   617.3  674.35   627.1  676.74   646.7  680.85   734.9  687.03   774.1   695.6
   842.7  701.08   881.8  708.95   911.2  712.28   940.6  719.23     970  731.74
   989.6  736.14  1058.2  758.43  1136.6  777.65  1175.8  790.62  1205.2   797.2
#Mann= 3 , 0 , 0
       0      .1       0   548.7    .045       0   627.1      .1       0
Bank Sta=548.7,627.1
XS Rating Curve= 0 ,0
Exp/Cntr=0.3,0.1

Type RM Length L Ch R = 1 ,38926   ,287.9,304.9,320.4
XS GIS Cut Line= 4
     1464057.546      255188.702     1464067.963       255693.91
      1464239.49      256101.285      1464569.88      256885.967
#Sta/Elev= 30
       0  828.28     311   771.9   408.1   743.6   417.9     739   427.6  732.21
   456.7  705.86   466.4  701.09   505.3  698.88   554.4   700.8   574.1  696.19
     633  676.36   662.5   673.9   701.8   673.9   711.6  675.52   750.9  689.81
   780.4  697.98   829.5  723.04   868.8  739.64     908  763.34   917.9  767.55
   966.9  779.88  1015.8  788.28  1064.8  801.05    1143  829.48  1280.1  854.03
  1348.6  862.22  1377.9  867.46  1554.1  909.34  1710.6  949.32  1798.7   967.2
#Mann= 3 , 0 , 0
       0      .1       0     633    .045       0   711.6      .1       0
Bank Sta=633,711.6
XS Rating Curve= 0 ,0
Exp/Cntr=0.3,0.1

Type RM Length L Ch R = 1 ,38621.1 ,407.8,435.5,462
XS GIS Cut Line= 3
     1464010.671      255183.493     1463897.137      255718.433
     1463554.255       256929.37
#Sta/Elev= 30
       0  825.32    68.4  812.21     166   787.3   283.2  750.36   380.8  732.27
   390.6  727.88   419.9  703.63   429.7  699.77   488.3  699.74   517.6  706.54
   537.1  707.03   576.4  698.19   625.5  692.39   656.8675.5747   674.7   671.9
   733.7  674.45   792.7  680.84   841.8  694.27     950  746.42   999.1  764.12
  1048.3  766.74  1136.8  745.94  1176.1  743.38    1186  746.16  1225.3  771.82
  1264.6  783.27  1353.1  823.19  1372.8  829.15  1687.4  879.39  1805.4  906.28
#Mann= 3 , 0 , 0
       0      .1       0   656.8    .045       0   733.7      .1       0
Bank Sta=656.8,733.7
XS Rating Curve= 0 ,0
Exp/Cntr=0.3,0.1

Type RM Length L Ch R = 1 ,38185.6 ,543.3,525.9,508
XS GIS Cut Line= 4
     1463988.283      255167.217     1463871.095      255557.842
     1463415.366      255592.565     1463063.804      255887.703
#Sta/Elev= 30
       0  823.32   165.1  782.29   223.3  760.89     301  736.42   349.6  722.81
   388.4  717.55   427.3  702.53   456.4   698.5   573.1  694.82   592.6  688.94
     612  677.72   621.8  673.01   631.5  670.63   641.2  670.59   660.7  674.41
     674 681.178   728.7  717.22   767.6  732.37   806.5  753.55   864.9  777.43
   933.2  801.82  1011.4  834.01  1030.9  835.14    1070  827.26  1099.3  818.16
  1138.3  814.29  1226.2  832.34  1245.8   838.8  1294.6  860.42  1323.9  866.94
#Mann= 3 , 0 , 0
       0      .1       0     612    .045       0     674      .1       0
Bank Sta=612,674
XS Rating Curve= 0 ,0
Exp/Cntr=0.3,0.1

Type RM Length L Ch R = 1 ,37659.7 ,713.1,694.4,675.5
XS GIS Cut Line= 2
      1463828.38       254756.41     1463177.338       255506.41
#Sta/Elev= 30
       0  890.56    88.5  858.23   157.3  831.66     177  822.48   226.2   796.5
   314.7   743.3   373.7  711.51   393.3  698.74   422.8  675.97   432.7   671.1
   442.5  669.81   452.3   669.7   481.8  669.98   491.7  670.93   550.7  681.91
     590  693.44   599.8  695.48   678.5  699.32   688.3  701.05   698.2  705.64
     708  712.56   717.8  721.24   737.5  740.82   786.7   764.2   865.3  803.29
   904.7  821.47     944  837.05   953.8  838.43   963.6  838.21   993.2  834.33
#Mann= 3 , 0 , 0
       0      .1       0   432.7    .045       0   491.7      .1       0
Bank Sta=432.7,491.7
XS Rating Curve= 0 ,0
Exp/Cntr=0.3,0.1

Type RM Length L Ch R = 1 ,36965.3 ,616.5,621.3,624.3
XS GIS Cut Line= 2
     1462807.546      254527.243     1462932.546      255579.327
#Sta/Elev= 30
       0  877.56    29.4  874.31      49  870.09   117.7  851.68   147.2  839.57
   176.6   824.5   235.4  787.68   333.5  729.35   441.4  672.87   451.3  670.25
   461.1   669.7   500.3  671.14   529.7  677.95   588.6  679.12   598.4  681.68
   627.8  695.64   637.6  697.78   657.3  698.02   667.1  700.58   706.3  720.54
   745.6   745.7     775  756.22   833.8  785.88   853.5  791.16   892.7  798.34
   902.5  798.31     981  789.67  1010.4  789.22    1030  790.74  1059.5  797.49
#Mann= 3 , 0 , 0
       0      .1       0   441.4    .045       0   500.3      .1       0
Bank Sta=441.4,500.3
XS Rating Curve= 0 ,0
Exp/Cntr=0.3,0.1

Type RM Length L Ch R = 1 ,36344   ,501.5,516.9,532.4
XS GIS Cut Line= 2
     1462302.338      254626.202     1462255.463      255719.952
#Sta/Elev= 30
       0   851.8    48.9  851.81      88  848.24   146.6  836.24   175.9  827.46
     215  810.43   254.1  780.88   322.6  740.52   371.4  707.31   381.2  701.91
   400.8  696.85   439.9  693.46   449.6  689.36   469.2   677.8   488.7  672.59
   508.3  669.94   527.8   669.7   566.9  669.74   586.5  671.76   615.8  679.75
   625.6  684.55   674.4  719.48   713.6  735.88     782  771.54   869.9  824.39
   889.5  834.42   918.8  844.82   957.9  852.79  1026.3   871.7  1094.8  883.06
#Mann= 3 , 0 , 0
       0      .1       0   488.7    .045       0   586.5      .1       0
Bank Sta=488.7,586.5
XS Rating Curve= 0 ,0
Exp/Cntr=0.3,0.1

Type RM Length L Ch R = 1 ,35827.2 ,480.8,501.2,519.4
XS GIS Cut Line= 3
     1462239.838      254615.785      1461953.38      254897.035
     1461312.755      255594.952
#Sta/Elev= 30
       0  830.09    19.6  827.01    78.3   804.9   146.9  784.16   195.8  762.14
     235  749.38   254.6  737.99     284  707.77   293.7  700.22   313.3  697.78
   430.8  696.84   450.3  692.12   489.4  676.05     587  667.36   616.3   665.7
   645.6  666.07   655.8669.1486   665.2  675.93     714  722.89   733.5  738.17
   792.1  769.85   811.6  776.11   840.9  774.06    1046   745.1  1085.1  735.42
  1133.9  716.38  1192.5   729.6  1212.1  743.25  1231.6   752.8  1348.8  789.18
#Mann= 3 , 0 , 0
       0      .1       0     587    .045       0   655.8      .1       0
Bank Sta=587,655.8
XS Rating Curve= 0 ,0
Exp/Cntr=0.3,0.1

Type RM Length L Ch R = 1 ,35326   ,223.4,221.9,220.9
XS GIS Cut Line= 2
     1462166.921      254636.618      1461390.88      254594.952
#Sta/Elev= 30
       0  789.95    19.7  778.17    39.4  768.78    68.9  756.86   157.4  724.06
   226.3  693.03   236.1  690.77   245.9  691.04   275.4  694.92   295.1  695.28
     305  694.43   314.8  692.31   324.6  688.65     364  670.22   373.8  666.97
   393.5  665.41   413.2  665.59     423  666.91   432.8  670.65     482  697.52
   550.9  738.68   570.6   752.9   609.9  786.17   629.6  800.89   649.3   812.7
     669  822.48   688.6  830.66   708.3  835.95     728  836.53   777.2  831.91
#Mann= 3 , 0 , 0
       0      .1       0     364    .045       0     423      .1       0
Bank Sta=364,423
XS Rating Curve= 0 ,0
Exp/Cntr=0.3,0.1

Type RM Length L Ch R = 1 ,35104.1 ,715.6,681,645.9
XS GIS Cut Line= 3
     1462224.213      254397.035     1461541.921      254407.452
      1461422.13      254527.243
#Sta/Elev= 30
       0  840.46     9.8  835.42    97.5  784.17     117  773.84   243.7  717.49
   331.4   675.3   360.7  665.73   370.4  664.23   385.1   663.9   409.4  664.06
   419.2  665.08   428.9  668.13   467.9  689.77   477.7  693.65   487.4  695.78
   565.4  697.02   604.4  698.98   623.9  701.55   633.6  704.78   643.4  709.58
   662.9  721.62   682.4  731.86   710.6  757.18   729.4  772.91   748.2  787.28
   757.7  793.15   785.9  807.66   804.7  815.32     833  823.88   851.8  827.18
#Mann= 3 , 0 , 0
       0      .1       0   360.7    .045       0   428.9      .1       0
Bank Sta=360.7,428.9
XS Rating Curve= 0 ,0
Exp/Cntr=0.3,0.1

Type RM Length L Ch R = 1 ,34423.1 ,727.8,721,713
XS GIS Cut Line= 2
     1461432.546      253501.202      1461422.13      254464.743
#Sta/Elev= 30
       0  866.66      59  874.99    88.5   878.2    98.3  878.32   108.2  876.88
   167.2  861.72   186.8   855.9   206.5  848.83   226.2  839.55   304.8   798.4
   393.3  745.38     413   731.7   432.6  716.28     472  687.97   491.6  669.47
   501.5  663.51   511.3  661.96   521.1  661.81   540.8  662.45   550.6  664.28
     590  674.45   619.5  688.92   629.3  691.43   806.3  701.21   816.1  704.56
   825.9   710.8   865.3  742.17   924.3  784.04   943.9  795.52   963.6  804.61
#Mann= 3 , 0 , 0
       0      .1       0   501.5    .045       0   550.6      .1       0
Bank Sta=501.5,550.6
XS Rating Curve= 0 ,0
Exp/Cntr=0.3,0.1

Type RM Length L Ch R = 1 ,33702.2 ,668.3,659.5,650.5
XS GIS Cut Line= 3
       1460559.5      253618.606     1460663.666      253962.356
     1460887.625      254649.856
#Sta/Elev= 30
       0  789.67    58.2  794.86   106.8  796.96   126.2  796.59   174.7  791.92
   300.9  773.12   310.6  771.01   359.2  752.95   456.9  705.16   525.3  674.47
   554.6  662.43   564.4  660.38   593.7  659.32   613.2  660.26     623   661.9
   652.3  667.28   662.1  671.09   701.2  691.34   710.9  693.79     750  698.48
   759.8  701.63     838  741.67   886.8  769.47   906.4  778.46   916.1  781.79
   935.7   786.1     965  796.23   974.8  797.08  1043.2   798.2  1082.2  801.04
#Mann= 3 , 0 , 0
       0      .1       0   554.6    .045       0     623      .1       0
Bank Sta=554.6,623
XS Rating Curve= 0 ,0
Exp/Cntr=0.3,0.1

Type RM Length L Ch R = 1 ,33042.7 ,607,608.4,609
XS GIS Cut Line= 2
     1459933.198      254211.054     1460618.961      255000.985
#Sta/Elev= 30
       0  772.22    58.7  774.06   146.6  772.75   156.4  770.95   166.2  765.95
     176  759.09   205.3  735.63   303.1  662.92   312.8  658.61   332.4   658.1
   371.5  658.54   381.3  660.64   400.8  667.93   410.6   669.4   469.3  673.87
   488.8   676.5   547.5  694.45   576.8  698.02   586.6  700.68   684.3  737.13
   762.6   772.8   772.3  776.28   791.9  780.34   801.7  783.73   860.3  808.56
     919  826.89   967.9  846.55   987.4  851.14    1007  853.99  1046.1   866.6
#Mann= 3 , 0 , 0
       0      .1       0   303.1    .045       0   381.3      .1       0
Bank Sta=303.1,381.3
XS Rating Curve= 0 ,0
Exp/Cntr=0.3,0.1

Type RM Length L Ch R = 1 ,32434.2 ,491,512.3,533.3
XS GIS Cut Line= 3
     1459575.559      254657.235     1460011.399      255198.734
     1460698.352      256534.405
#Sta/Elev= 30
       0  754.17    78.3  748.37   137.1  731.79   254.6  690.17   323.1  676.38
   362.2  657.11   381.8   656.3   421.1658.2568   450.4     666   499.3  695.07
   548.3  704.29     607  745.88   636.4  762.52   665.7  777.53   763.8  818.26
   822.7  833.99   911.1  846.75  1048.5  879.64  1097.6   895.7  1323.4  888.82
  1372.5     890  1411.7  884.16  1470.6  888.65  1509.9  880.68    1559  902.72
  1598.3  915.87    1824  959.47  1971.3  1003.1  2069.5  1005.9  2197.1 1001.89
#Mann= 3 , 0 , 0
       0      .1       0   362.2    .045       0   421.1      .1       0
Bank Sta=362.2,421.1
XS Rating Curve= 0 ,0
Exp/Cntr=0.3,0.1

Type RM Length L Ch R = 1 ,31921.9 ,373.6,378.5,382.6
XS GIS Cut Line= 3
     1459513.059      254667.651     1459307.267      255438.499
     1458059.463      256647.252
#Sta/Elev= 30
       0  749.45   126.5  737.42   262.7  695.83   321.1  682.71     360   665.7
   447.6   657.8   486.5   656.2   510.1660.4938   583.8  718.58   671.4  754.45
   739.5  766.14   768.7  775.97   846.9  790.75    1004  830.32  1072.7  844.22
    1161  855.83  1229.7  868.33  1396.6  912.01  1465.3  919.88  1671.4  933.31
  1779.4  931.89  1877.5  937.66  1965.8  936.07  2113.1  939.42  2230.8  954.09
  2309.4  973.25  2378.1  997.12  2407.5 1004.24  2476.2 1015.91  2535.1 1018.74
#Mann= 3 , 0 , 0
       0      .1       0   447.6    .045       0   510.1      .1       0
Bank Sta=447.6,510.1
XS Rating Curve= 0 ,0
Exp/Cntr=0.3,0.1
